--- RIGHTBFLCK.prj (project) ---

Proj Title=RIGHTBFLCK
Current Plan=p01
Default Exp/Contr=0,0
English Units
Geom File=g01
Flow File=f01
Plan File=p01
BEGIN DESCRIPTION:
END DESCRIPTION:
DSS Export Rating Curves= 0
DSS Export Rating Curve Sorted= 0
DSS Export Volume Flow Curves= 0
DXF OffsetX= 0
DXF OffsetY= 0
DXF ScaleX= 0
DXF ScaleY= 0

--- RIGHTBFLCK.p01 (plan) ---

Plan Title=Floodplain
Program Version=4.00
Geom File=g01
Flow File=f01
K Sum by GR=0
Std Step Tol=0.01
Critical Tol=0.01
Num of Std Step Trials=20
Max Error Tol=0.3
Flow Tol Ratio=0.001
Split Flow NTrial=30
Split Flow Tol=0.02
Split Flow Ratio=0.02
Log Output Level=0
Friction Slope Method=1
Unsteady Friction Slope Method=2
Unsteady Bridges Friction Slope Method=1
Global Log Level=0
CheckData=False
Run HTab=0
Run UNet=0
Run PostProcess=0
UNET Theta=0
UNET Theta Warmup=0
UNET ZTol=0
UNET ZSATol=0
UNET MxIter=0
UNET MaxInSteps=0
UNET DtIC=0
UNET DtMin=0
UNET MaxCRTS=0
UNET WFStab=0
UNET SFStab=0
UNET WFX=0
UNET SFX=0
UNET DSS MLevel=0
UNET DZMax Abort=0
UNET Convert EG Bridges=0
UNET Use Existing IB Tables=0
UNET Froude Limit=0
UNET Froude Power=0
Write IC File=0
Echo Input=False
Echo Output=False
Write Detailed=0

--- RIGHTBFLCK.f01 (steady flow) ---

Flow Title=NFF Regression Equation
Program Version=4.10
Number of Profiles= 1
Profile Names=P100yr
River Rch & RM=RIGHTBFLCK,Main            ,20665.7
944.7448
River Rch & RM=RIGHTBFLCK,Main            ,20265.3
967.8691
River Rch & RM=RIGHTBFLCK,Main            ,17093.5
1063.337
River Rch & RM=RIGHTBFLCK,Main            ,14653.8
1173.221
River Rch & RM=RIGHTBFLCK,Main            ,11967.8
1255.626
River Rch & RM=RIGHTBFLCK,Main            ,11511.1
1479.372
River Rch & RM=RIGHTBFLCK,Main            ,9118.2
1546.518
River Rch & RM=RIGHTBFLCK,Main            ,6309.8
1716.204
River Rch & RM=RIGHTBFLCK,Main            ,5504.9
1873.951
River Rch & RM=RIGHTBFLCK,Main            ,4784.1
1931.974
Boundary for River Rch & Prof#=RIGHTBFLCK,Main            , 1
Up Type= 0
Dn Type= 1
Dn Known WS=1013.31
DSS Import GetInterval= 0
DSS Import GetPeak= 0
DSS Import FillOption= 0

--- RIGHTBFLCK.g01 (geometry) ---

Geom Title=USGS 10m DEM
Program Version=4.10

River Reach=RIGHTBFLCK      ,Main
Reach XY= 30
      1751676.81      282419.495      1749924.17      282527.822
     1748871.643      282711.362     1748562.221      282627.125
     1748064.216      282679.097     1747803.632      282572.161
     1747426.746      282614.284     1746553.354      282414.987
     1746197.433      282235.181     1745698.613      281736.361
     1745014.826      279570.315     1744736.858       279083.87
     1744153.123       278619.43     1743848.516      278570.786
     1743744.277      278415.587     1743016.926      277916.401
     1742143.641      277670.862     1741642.139      277405.633
     1740935.635      276605.315     1740683.047      276494.844
     1740409.943      276149.809     1740011.106      275979.631
      1739811.02      275738.979     1739129.996      275798.047
     1738671.348      275517.762     1737994.957      275401.942
     1737502.721      275070.696     1736536.779      275176.092
     1735427.221      275054.481     1734919.928      275194.624

Type RM Length L Ch R = 1 ,20665.7 ,402.8,400.4,397.9
XS GIS Cut Line= 2
     1751670.077       282206.01     1751664.189      282653.197
#Sta/Elev= 30
       0 1542.14    19.4 1529.77    48.6 1511.86    58.3 1507.34    68.1  1504.7
    77.8 1504.36   145.8 1484.54   155.6 1484.48   184.7 1474.22   194.4 1471.54
   204.2 1471.16   204.8 1471.33   213.9 1473.89   219.8 1476.96   223.6 1478.93
   233.3 1479.29   252.8 1489.23   272.2 1498.54     282 1504.04   301.4 1516.52
   311.1 1517.62   320.8 1523.19     350  1543.4   379.2 1562.93   388.9 1564.71
   398.6 1569.86   418.1 1584.23   427.8 1590.64   437.5 1596.14   447.2 1600.97
#Mann= 3 , 0 , 0
       0     .08       0   204.8    .045       0   219.8     .08       0
Bank Sta=204.8,219.8
XS Rating Curve= 0 ,0
Exp/Cntr=0.3,0.1

Type RM Length L Ch R = 1 ,20265.3 ,396.6,400,403.4
XS GIS Cut Line= 2
     1751247.462      282224.384      1751292.15      282692.103
#Sta/Elev= 30
       0  1523.5    29.4 1507.44    39.2 1507.21    58.7 1495.99    68.5 1491.24
    78.3 1488.48   107.7 1481.92   117.5 1481.86   146.8 1475.19     186 1465.42
   195.8 1465.16   215.4 1459.99   220.5 1459.86   225.1 1459.75   234.9 1465.06
   235.5 1465.71   254.5 1486.12   264.3 1495.81   274.1 1497.72   283.9 1505.36
   293.7 1514.26   303.4  1522.5   342.6 1551.39   352.4 1553.52   362.2 1558.65
   381.8 1571.76   420.9 1596.15   430.7 1598.14   440.5 1602.41   469.8 1624.09
#Mann= 3 , 0 , 0
       0     .08       0   220.5    .045       0   235.5     .08       0
Bank Sta=220.5,235.5
XS Rating Curve= 0 ,0
Exp/Cntr=0.3,0.1

Type RM Length L Ch R = 1 ,19865.3 ,392.4,389.7,387
XS GIS Cut Line= 2
     1750882.809      282240.239     1750854.641      282737.855
#Sta/Elev= 30
       0 1509.67     9.8    1505    39.1 1486.09    48.9 1481.21    58.6  1478.3
    68.4 1476.45      88 1474.67     127 1466.34   146.6 1461.48   166.1 1458.96
   205.2 1448.72     215  1446.8   220.6 1447.95   235.6 1452.03   244.3 1456.68
   263.9 1477.09   273.6 1485.89   283.4 1493.84     303  1508.2   312.7 1512.28
   322.5 1515.06     342 1527.94   381.1 1551.47   390.9 1555.39   400.7 1557.49
   439.8  1581.8   459.3 1595.19   469.1 1600.24   478.9 1602.19   498.4  1616.2
#Mann= 3 , 0 , 0
       0     .08       0   220.6    .045       0   235.6     .08       0
Bank Sta=220.6,235.6
XS Rating Curve= 0 ,0
Exp/Cntr=0.3,0.1

Type RM Length L Ch R = 1 ,19475.6 ,408.8,408.5,408.1
XS GIS Cut Line= 2
     1750467.703      282258.287     1750500.752      282774.864
#Sta/Elev= 30
       0 1495.01    19.5 1478.38    29.3 1474.25    39.1 1470.76    48.8 1465.57
    58.6  1463.3    97.7 1457.75   117.2 1456.25     127 1454.72   146.5 1451.39
   175.8 1445.43   185.6  1444.1   195.3 1443.39   214.9 1439.12   219.3 1438.82
   224.6 1438.46   234.3 1440.84   244.2 1446.98   253.9 1454.14   263.7 1458.96
   273.5 1460.72   302.8  1480.8   341.8 1508.38   361.4 1516.94   400.4 1548.39
   429.7 1573.63   439.5 1574.53   478.6 1613.47   507.9 1643.89   517.6 1644.01
#Mann= 3 , 0 , 0
       0     .08       0   219.3    .045       0   234.3     .08       0
Bank Sta=219.3,234.3
XS Rating Curve= 0 ,0
Exp/Cntr=0.3,0.1

Type RM Length L Ch R = 1 ,19067.1 ,484.4,483.7,483.1
XS GIS Cut Line= 2
     1750057.825      282276.108     1750099.955      282816.777
#Sta/Elev= 30
       0 1484.71    38.7 1467.88    58.1 1460.22    67.8 1457.28    77.5 1456.64
    96.8 1449.93   135.6 1439.58   145.3  1437.3     155 1437.27   164.6 1435.86
   222.7 1429.75   234.7 1429.48   242.1 1428.95   249.7    1429   261.5 1430.93
   300.2 1440.25   309.9 1440.98   319.6 1444.25   329.3 1449.79   377.7 1479.65
   387.4 1482.25     397 1486.13   426.1 1507.77   455.2 1527.26   474.5 1534.38
   493.9 1550.22   503.6 1557.01   513.3 1564.56   532.6    1581   542.3 1587.04
#Mann= 3 , 0 , 0
       0     .08       0   234.7    .045       0   249.7     .08       0
Bank Sta=234.7,249.7
XS Rating Curve= 0 ,0
Exp/Cntr=0.3,0.1

Type RM Length L Ch R = 1 ,18583.3 ,364.2,362.6,360.9
XS GIS Cut Line= 2
      1749567.55      282297.424     1749630.709      282865.848
#Sta/Elev= 30
       0 1475.42     9.7 1469.46    29.1 1463.67    48.5 1454.19    87.2    1439
    96.9 1436.39   106.6 1435.35   135.7 1425.44   155.1 1420.29   203.6 1415.46
   213.3 1416.26   232.6  1423.3   242.3 1425.43     252 1423.34   261.7 1423.29
   271.4  1420.2   285.2 1418.19   300.2 1417.98   310.2 1420.32   319.9 1427.55
   329.6 1436.82   339.3 1439.14     349 1446.17     378 1471.19   407.1 1493.45
   426.5  1501.2   494.4 1555.82   504.1  1560.9   513.8 1564.45   571.9 1615.66
#Mann= 3 , 0 , 0
       0     .08       0   285.2    .045       0   300.2     .08       0
#XS Ineff= 2 , 0
          242.61 1424.31
Permanent Ineff=
       F       F
Bank Sta=285.2,300.2
XS Rating Curve= 0 ,0
Exp/Cntr=0.3,0.1

Type RM Length L Ch R = 1 ,18220.7 ,57.1,57.1,57.1
XS GIS Cut Line= 2
     1749183.919      282322.763     1749289.848      282901.494
#Sta/Elev= 30
       0 1477.01    19.6 1462.66      49 1442.97    58.8 1442.94    78.4 1432.08
   117.7 1411.94   127.5 1409.79   147.1 1408.74   205.9 1402.47   225.5 1402.06
   235.3 1403.68   274.6 1418.98   284.4 1421.45   294.2    1422     304 1421.18
   323.6 1417.38   333.4 1416.76   342.7 1419.01   357.7 1426.24   372.6 1432.52
   382.4 1434.68   411.8 1458.71   421.6 1465.73   441.3 1476.28   451.1    1480
   460.9 1481.68   470.7 1484.94   539.3 1512.96   549.1  1513.6   588.4 1530.21
#Mann= 3 , 0 , 0
       0     .08       0   342.7    .045       0   357.7     .08       0
#XS Ineff= 2 , 0
          294.85 1421.39
Permanent Ineff=
       F       F
Bank Sta=342.7,357.7
XS Rating Curve= 0 ,0
Exp/Cntr=0.3,0.1

Type RM Length L Ch R = 1 ,18163.5 ,335,345.4,355.8
XS GIS Cut Line= 2
     1749127.277      282329.746     1749233.016      282907.437
#Sta/Elev= 30
       0 1467.75    29.4  1446.7    39.2 1444.84    48.9 1440.48    78.3 1423.86
   107.7 1411.65   117.5 1408.82   205.6 1400.08   215.3 1400.32   225.1 1401.88
   264.3 1418.63   274.1 1420.03   283.9 1418.02   293.6  1417.8   303.4 1414.34
   313.2  1412.5   332.8 1411.88   341.4  1412.8   352.4 1417.33   356.4  1420.3
   362.2 1424.61     372 1425.41   420.9 1461.62   430.7  1467.6   440.5  1470.3
     460 1471.99   469.8 1474.65   518.8 1495.06   538.4 1498.29   587.3 1515.11
#Mann= 3 , 0 , 0
       0     .08       0   341.4    .045       0   356.4     .08       0
#XS Ineff= 2 , 0
          274.23 1419.76
Permanent Ineff=
       F       F
Bank Sta=341.4,356.4
XS Rating Curve= 0 ,0
Exp/Cntr=0.3,0.1

Type RM Length L Ch R = 1 ,17818.2 ,352.9,347,341.1
XS GIS Cut Line= 4
     1748820.478      282374.645     1748857.619      282671.172
     1748834.667      282751.504     1748851.061      282933.481
#Sta/Elev= 30
       0  1450.1    19.3    1440    48.2  1426.7    57.8 1423.27    67.5 1422.64
   125.3 1399.68     135 1397.45   231.4  1394.4     241 1395.13   250.6 1397.53
   260.3 1401.39   279.6 1411.43   289.2  1413.8   298.8 1414.16   308.1 1413.02
   317.4 1410.26   327.9 1408.86     336  1412.4   342.9 1417.13   354.5 1421.59
   382.4 1423.26   411.2 1422.89   420.9 1426.44   430.5 1433.07   449.7 1448.84
   468.9 1457.73   526.6 1512.34   536.2 1519.98   545.9 1521.72   565.1 1540.42
#Mann= 3 , 0 , 0
       0     .08       0   327.9    .045       0   342.9     .08       0
#XS Ineff= 2 , 0
          292.02 1413.93
Permanent Ineff=
       F       F
Bank Sta=327.9,342.9
XS Rating Curve= 0 ,0
Exp/Cntr=0.3,0.1

Type RM Length L Ch R = 1 ,17471.1 ,377.5,377.6,377.6
XS GIS Cut Line= 2
     1748517.182      282404.963     1748506.443      282983.419
#Sta/Elev= 30
       0 1442.57    19.6 1437.22    39.2 1427.42    78.4 1410.86    98.1 1406.78
   137.3 1390.36   156.9 1385.87   176.5 1384.04   213.2 1377.18   215.7 1376.75
   225.5 1376.83   228.2 1377.83   245.2 1384.54     255 1386.55   274.6 1397.71
   313.8 1416.96   323.6 1420.47   333.4 1422.03   372.6 1445.02   392.2 1460.12
     402 1465.83   411.8 1467.78   431.5 1482.14   470.7 1506.86   480.5 1511.84
   490.3 1513.44   549.1 1552.88   558.9 1557.77   568.8 1558.98   578.6 1564.81
#Mann= 3 , 0 , 0
       0     .08       0   213.2    .045       0   228.2     .08       0
Bank Sta=213.2,228.2
XS Rating Curve= 0 ,0
Exp/Cntr=0.3,0.1

Type RM Length L Ch R = 1 ,17093.5 ,397.7,395.4,393.2
XS GIS Cut Line= 2
     1748150.162       282420.88      1748145.04      282965.863
#Sta/Elev= 30
       0 1434.31    19.5 1424.31    48.7 1411.18    58.4 1411.11   107.1 1388.02
   126.5 1380.07   136.2 1379.69   155.7 1376.38   204.4 1370.29   214.1 1370.06
   245.2 1366.58     253 1366.48   260.2 1367.92   262.8 1368.44   282.2 1377.39
     292 1378.62   301.7 1382.21   340.6 1402.38   350.4 1409.65   360.1 1418.16
   369.8 1421.46   379.6 1426.89   408.8 1453.48     438 1478.98   457.4 1486.85
   486.6    1509   515.8 1533.18   525.5 1537.72   535.3  1541.2     545 1549.16
#Mann= 3 , 0 , 0
       0     .08       0   245.2    .045       0   260.2     .08       0
Bank Sta=245.2,260.2
XS Rating Curve= 0 ,0
Exp/Cntr=0.3,0.1

Type RM Length L Ch R = 1 ,16698   ,384.1,390.5,396.9
XS GIS Cut Line= 2
     1747764.106      282384.112     1747800.477      282911.459
#Sta/Elev= 30
       0 1418.59     9.8 1410.28    19.6 1402.65    29.4 1396.12    39.2 1390.88
    48.9 1386.82    58.7  1383.4    68.5 1380.97    78.3  1380.2   127.3 1364.98
   146.8 1361.52   156.6 1361.16     181 1356.37     186 1355.57     196 1355.76
   205.6 1358.55   215.4 1363.38   225.1 1367.06   234.9 1367.58   303.4 1394.26
   313.2 1394.56     323 1399.08   362.2 1419.08   381.8 1429.76   391.6 1429.76
   420.9 1449.23   460.1 1477.48   469.9  1477.9   479.6 1484.98   528.6 1523.84
#Mann= 3 , 0 , 0
       0     .08       0     181    .045       0     196     .08       0
Bank Sta=181,196
XS Rating Curve= 0 ,0
Exp/Cntr=0.3,0.1

Type RM Length L Ch R = 1 ,16307.5 ,378,377.3,376.6
XS GIS Cut Line= 2
      1747447.11      282353.922      1747342.27       282839.11
#Sta/Elev= 30
       0 1398.45     9.7  1397.1    29.2 1387.16    68.1 1368.79    77.9 1365.64
    87.6 1364.12   107.1 1357.87   116.8 1355.54     146 1352.09   165.5  1351.1
   223.9 1345.52   243.3 1344.36   251.8 1343.42   262.8 1343.05   266.8 1344.18
   272.5  1345.8   282.3  1353.4     292 1362.07   301.7  1369.8   311.5 1376.26
   321.2 1378.08   350.4 1401.38   389.3 1435.25   399.1 1436.46   408.8    1444
   428.2 1461.01   467.2 1493.58   476.9 1496.85   486.6 1501.81   496.4 1509.94
#Mann= 3 , 0 , 0
       0     .08       0   251.8    .045       0   266.8     .08       0
Bank Sta=251.8,266.8
XS Rating Curve= 0 ,0
Exp/Cntr=0.3,0.1

Type RM Length L Ch R = 1 ,15929.9 ,416.5,419.8,423.1
XS GIS Cut Line= 2
     1747071.644      282294.001     1746982.885      282782.365
#Sta/Elev= 30
       0 1372.23     9.7 1366.44    19.5 1362.15    29.2 1359.39    38.9 1359.14
    48.7 1357.42    77.9 1353.76   107.1 1349.17   116.8 1348.91   175.2 1340.68
   204.4 1340.48   214.1 1338.23   222.4 1335.65   223.8 1335.21   233.6 1335.09
   237.4 1337.03   243.3 1340.03     253 1347.91   262.8  1355.3   272.5 1359.33
   282.2 1361.93   340.6 1402.86   350.4 1408.66   360.1 1409.67   389.3 1431.27
   418.5 1452.27   428.2 1459.63     438 1459.73   447.7 1466.91   496.4 1505.27
#Mann= 3 , 0 , 0
       0     .08       0   222.4    .045       0   237.4     .08       0
Bank Sta=222.4,237.4
XS Rating Curve= 0 ,0
Exp/Cntr=0.3,0.1

Type RM Length L Ch R = 1 ,15509.9 ,402.6,407,411.4
XS GIS Cut Line= 2
     1746733.991      282107.403     1746534.988      282694.705
#Sta/Elev= 30
       0 1392.78    38.8 1378.45    48.4 1377.46    58.1 1374.25   116.3 1352.05
     155 1342.58   174.4 1341.18   193.8 1338.44   300.4 1330.32   346.5 1324.76
   348.8 1324.52   358.5  1324.9   361.5 1326.25   377.9  1332.2   387.6 1336.89
   426.3  1366.9   445.7 1379.35   455.4 1384.77   465.1 1385.24   494.1  1401.6
   513.5 1416.93   532.9 1434.47   542.6 1439.62   552.3 1443.02     562 1451.52
   571.7 1458.43   581.4 1462.84     591 1464.29   610.4 1465.44   620.1 1463.68
#Mann= 3 , 0 , 0
       0     .08       0   346.5    .045       0   361.5     .08       0
Bank Sta=346.5,361.5
XS Rating Curve= 0 ,0
Exp/Cntr=0.3,0.1

Type RM Length L Ch R = 1 ,15102.8 ,441.6,448.5,455.6
XS GIS Cut Line= 2
     1746446.058      281959.021     1746100.304      282545.998
#Sta/Elev= 30
       0 1402.63     9.7 1395.54    19.5 1394.01    29.2 1388.08    58.4 1367.14
    97.3 1342.52   116.8 1338.11   126.5 1334.27     146 1327.98   155.7 1327.22
   223.8    1327   301.7 1325.07   354.1 1318.06   360.1 1317.55   369.1 1319.31
   389.3 1325.54     399 1333.14   428.2 1351.08   447.7 1362.47   457.4 1366.59
   467.1 1367.92   476.9 1371.26     545 1390.26   564.5 1394.35   583.9 1401.77
   613.1    1415   632.6 1424.77   642.3 1431.63     652 1436.28   681.2  1455.9
#Mann= 3 , 0 , 0
       0     .08       0   354.1    .045       0   369.1     .08       0
Bank Sta=354.1,369.1
XS Rating Curve= 0 ,0
Exp/Cntr=0.3,0.1

Type RM Length L Ch R = 1 ,14653.8 ,340.6,345.7,350.7
XS GIS Cut Line= 2
     1746145.552      281782.169     1745680.636      282208.339
#Sta/Elev= 30
       0 1386.48    19.4 1374.87    29.1 1373.32    58.2 1356.98      97  1336.9
   116.4 1323.44   126.1 1318.31   135.8 1315.54   155.2 1313.54   232.9 1313.01
     262 1310.95   298.6 1306.51   310.5  1306.1   313.6 1306.99   320.2  1308.9
   329.9 1316.59   349.3 1333.43     359 1335.66   368.7 1340.93   407.5 1367.11
   417.2 1371.38   446.3 1379.97   465.7 1387.28   475.4 1388.83   485.1 1391.71
   533.7 1413.23   572.5 1428.36   582.2 1435.38   591.9    1445   630.7 1471.82
#Mann= 3 , 0 , 0
       0     .08       0   298.6    .045       0   313.6     .08       0
Bank Sta=298.6,313.6
XS Rating Curve= 0 ,0
Exp/Cntr=0.3,0.1

Type RM Length L Ch R = 1 ,14308   ,394.6,396.4,398.3
XS GIS Cut Line= 2
     1745964.834      281588.065     1745524.416      281833.089
#Sta/Elev= 30
       0 1399.86     9.7  1394.1    19.4 1382.67    29.1 1369.58    48.5 1339.28
    58.2 1327.56    67.8 1321.51    77.5 1319.66    96.9 1317.06   116.3 1313.68
   135.7 1308.85   145.4 1307.47   193.8 1304.58   222.9 1303.56   232.6  1302.3
   297.2 1296.03   300.4 1295.79   310.2 1297.41   312.2 1298.57   319.8 1302.99
   329.5 1312.99   339.2 1322.42     378 1346.04   387.7 1349.36   397.4 1354.89
   416.8 1366.92   426.4 1373.24   436.1 1382.71   474.9 1399.96     504 1413.52
#Mann= 3 , 0 , 0
       0     .08       0   297.2    .045       0   312.2     .08       0
Bank Sta=297.2,312.2
XS Rating Curve= 0 ,0
Exp/Cntr=0.3,0.1

Type RM Length L Ch R = 1 ,13911.1 ,396.2,399.9,403.6
XS GIS Cut Line= 2
     1745773.831      281269.514     1745347.851      281463.142
#Sta/Elev= 30
       0 1316.01     9.8 1310.91    19.5 1308.27    48.7 1302.83    58.5 1299.87
     117 1290.72   126.7    1290   136.5  1290.2   175.5 1293.01   185.2 1293.29
     195 1292.28   204.7 1290.06   224.2 1284.27     226 1283.95     234 1282.52
     241 1282.79   243.7 1282.89   253.5 1285.83   263.2 1288.16   321.7 1301.34
   341.2 1306.51   350.9 1309.69   360.7  1316.1   399.7 1333.31   409.4 1338.43
   428.9 1349.47   438.7 1354.48   448.4 1360.64   458.2 1371.91   467.9 1377.39
#Mann= 3 , 0 , 0
       0     .08       0     226    .045       0     241     .08       0
Bank Sta=226,241
XS Rating Curve= 0 ,0
Exp/Cntr=0.3,0.1

Type RM Length L Ch R = 1 ,13511.1 ,399.7,400,400.2
XS GIS Cut Line= 2
     1745667.843      280927.324     1745157.551      281064.418
#Sta/Elev= 30
       0 1355.88    39.1 1320.48    48.9 1312.48    58.7 1306.46    68.5  1301.1
     137 1281.07   146.8 1279.66   156.6 1279.61   176.1 1281.32   185.9 1281.94
   195.7  1282.1   205.5 1281.47   234.8 1278.34   244.6 1277.18     257 1275.21
   264.2 1274.34     272 1275.73     274 1276.09   283.8  1280.5   293.6 1285.92
   303.3 1290.68   322.9 1299.38   352.3 1312.99     362 1321.48   401.2 1340.54
     411 1344.79   440.3  1356.5   459.9 1368.28   489.2  1380.1   528.4 1394.58
#Mann= 3 , 0 , 0
       0     .08       0     257    .045       0     272     .08       0
#XS Ineff= 2 , 0
          197.94 1282.11
Permanent Ineff=
       F       F
Bank Sta=257,272
XS Rating Curve= 0 ,0
Exp/Cntr=0.3,0.1

Type RM Length L Ch R = 1 ,13111.1 ,401.4,400,398.5
XS GIS Cut Line= 2
      1745550.62      280548.863     1745039.989      280679.709
#Sta/Elev= 30
       0 1337.72    29.3 1316.55      39 1309.85    48.8 1303.96    68.3 1294.52
    78.1 1286.69    87.8 1281.63    97.6 1277.51   107.4 1274.36   117.1 1272.98
   146.4 1272.74     166 1271.85   185.5 1269.22   225.8 1265.37   234.3 1264.82
   240.8 1264.98     244 1265.06   253.8 1267.32   263.6 1271.53   273.3 1277.44
   302.6 1289.96   322.1 1299.22   361.2 1312.92   370.9 1321.49   380.7 1328.07
     449 1371.17   458.8 1380.17   468.6 1388.41   488.1 1396.23   527.1 1412.92
#Mann= 3 , 0 , 0
       0     .08       0   225.8    .045       0   240.8     .08       0
Bank Sta=225.8,240.8
XS Rating Curve= 0 ,0
Exp/Cntr=0.3,0.1

Type RM Length L Ch R = 1 ,12711.1 ,397,399.9,402.8
XS GIS Cut Line= 2
     1745428.586      280154.865     1744941.207      280312.804
#Sta/Elev= 30
       0 1305.13     9.7 1298.52    19.3  1292.7      29 1287.81    38.7 1283.74
    48.3 1280.49      58 1277.62    67.7 1274.98      87 1270.41    96.7 1267.03
   125.7 1261.36   135.3 1260.27   193.3 1256.73   229.9 1255.47     232 1255.42
   241.7 1256.23   244.9 1257.58   251.3 1260.29     261 1267.46   270.7    1273
     290  1287.3   328.7 1308.24   367.3 1328.51     377 1334.23   386.7  1343.5
     464 1382.49   483.3 1396.79     493 1401.11   502.7 1404.84   512.3 1407.81
#Mann= 3 , 0 , 0
       0     .08       0   229.9    .045       0   244.9     .08       0
Bank Sta=229.9,244.9
XS Rating Curve= 0 ,0
Exp/Cntr=0.3,0.1

Type RM Length L Ch R = 1 ,12311.1 ,349.2,343.2,337.3
XS GIS Cut Line= 2
      1745353.75      279800.736      1744829.51      279897.931
#Sta/Elev= 30
       0 1321.02    29.1 1302.85    38.8 1295.77    48.5  1285.8    58.2 1282.07
   135.7 1258.52   145.4 1254.06   155.1  1252.6     223 1248.95   242.4 1247.43
     280 1245.29   290.8 1245.01     295 1246.15   300.5 1247.64   310.2 1255.39
   329.6 1274.88   339.3 1287.48   358.7 1302.24   378.1 1316.59   416.8 1344.18
   426.5  1355.7   436.2 1362.27   445.9 1368.22   465.3 1379.47   484.7 1389.78
   494.4 1394.48   504.1 1398.78   513.8 1403.88   523.5 1414.88   533.2 1425.16
#Mann= 3 , 0 , 0
       0     .08       0     280    .045       0     295     .08       0
Bank Sta=280,295
XS Rating Curve= 0 ,0
Exp/Cntr=0.3,0.1

Type RM Length L Ch R = 1 ,11967.8 ,462.5,456.6,450.7
XS GIS Cut Line= 2
     1745384.668      279333.329     1744697.744      279664.021
#Sta/Elev= 30
       0 1299.44    29.3 1302.57    78.2 1311.84      88 1312.65   107.5  1310.4
   117.3 1308.85   127.1 1302.48   185.7 1279.86     215 1266.29   224.8 1258.82
   234.6  1255.1   332.3 1244.54   420.3 1241.21     434 1238.94     449 1237.25
   449.6 1237.21   459.4 1238.84   469.2 1244.73   488.7 1261.79     518 1282.68
   537.6 1301.45   576.7 1328.15     606 1342.67   615.8 1349.02   635.3 1366.31
   645.1 1372.39     694 1400.42   733.1 1417.98   742.8 1423.93   762.4 1430.25
#Mann= 3 , 0 , 0
       0     .08       0     434    .045       0     449     .08       0
Bank Sta=434,449
XS Rating Curve= 0 ,0
Exp/Cntr=0.3,0.1

Type RM Length L Ch R = 1 ,11511.1 ,396.7,389.5,382.3
XS GIS Cut Line= 2
     1745042.721      278900.867     1744488.381      279376.147
#Sta/Elev= 30
       0  1342.7    19.5    1325    77.9 1285.55   107.1 1271.51   116.8 1265.18
   136.3 1248.95   155.8 1239.15     185 1233.45   243.4 1230.08   321.3 1237.08
     331 1237.06   346.8 1231.35   350.5 1229.41   360.2 1228.65   361.8 1229.17
   428.4 1258.32   438.1  1259.1   467.3 1270.43   486.8 1284.18   506.3 1293.91
     516 1297.22   535.5 1301.78     555 1309.01   584.2 1314.63   603.6 1320.33
   642.6 1323.66     662 1327.48     701 1338.98   710.7 1344.71   730.2 1351.08
#Mann= 3 , 0 , 0
       0     .08       0   346.8    .045       0   361.8     .08       0
#XS Ineff= 2 , 0
          325.32 1237.11
Permanent Ineff=
       F       F
Bank Sta=346.8,361.8
XS Rating Curve= 0 ,0
Exp/Cntr=0.3,0.1

Type RM Length L Ch R = 1 ,11121.6 ,265.1,270,274.8
XS GIS Cut Line= 2
     1744666.194      278566.998     1744317.957      279141.814
#Sta/Elev= 30
       0 1380.95    48.7 1347.03    68.2 1331.78    77.9 1326.77    87.7 1319.83
   146.1 1277.36   155.8 1274.56   175.3 1258.21   204.5 1229.15   214.3 1222.24
     224 1220.07   253.2 1220.73   292.2 1221.97   321.4 1225.14   360.4 1226.76
   370.1 1225.51   378.5 1222.67   389.6  1219.5   393.5 1219.68   418.8 1223.46
   438.3 1224.95   457.8 1229.76   467.5 1233.31   506.5 1254.74     526 1260.78
   545.4 1273.96   584.4 1295.39   594.2 1300.18   603.9 1300.94   672.1 1338.68
#Mann= 3 , 0 , 0
       0     .08       0   378.5    .045       0   393.5     .08       0
#XS Ineff= 2 , 0
          358.42 1226.69
Permanent Ineff=
       F       F
Bank Sta=378.5,393.5
XS Rating Curve= 0 ,0
Exp/Cntr=0.3,0.1

Type RM Length L Ch R = 1 ,10851.6 ,541.4,540.7,540
XS GIS Cut Line= 2
     1744516.964      278455.075     1744065.423       278930.38
#Sta/Elev= 30
       0 1352.82     9.8 1349.72    19.6 1343.48    97.8 1287.39   107.6 1284.89
   127.2 1267.05   166.3 1239.74   195.7 1220.37   205.5 1216.13   215.3 1214.98
     225 1214.54   264.2 1215.61   293.6 1215.83   352.3 1219.34     362 1219.24
   371.8 1216.66   376.9 1214.67   381.6 1212.83   391.4 1212.31   391.9 1212.44
   420.8  1220.4   430.5  1223.6   489.2 1236.96   508.8 1243.22   538.2 1248.14
   567.5 1255.15   606.7 1266.71   626.2 1272.86     636 1276.61   655.6 1281.91
#Mann= 3 , 0 , 0
       0     .08       0   376.9    .045       0   391.9     .08       0
#XS Ineff= 2 , 0
          357.62 1219.25
Permanent Ineff=
       F       F
Bank Sta=376.9,391.9
XS Rating Curve= 0 ,0
Exp/Cntr=0.3,0.1

Type RM Length L Ch R = 1 ,10310.6 ,441,438.9,436.6
XS GIS Cut Line= 2
     1744135.942      278196.974     1743687.001      278672.843
#Sta/Elev= 30
       0  1345.8     9.8 1339.32    29.3 1322.29    87.9 1281.69    97.6 1275.21
   107.4 1272.62   117.2 1266.01   136.7 1250.05   146.5 1241.13   156.2 1230.62
   175.8 1216.08   185.5 1210.36   195.3 1208.04   283.2 1207.75   312.5 1208.09
   390.6  1211.7   400.3 1210.51   410.1 1207.06   429.6 1202.61   439.4  1202.1
   452.3 1203.63   467.3  1208.2     498 1217.25   517.5 1224.35   527.3 1225.84
   556.6 1242.77   605.4 1273.88   615.2 1277.39   624.9 1279.12   654.2 1297.23
#Mann= 3 , 0 , 0
       0     .08       0   452.3    .045       0   467.3     .08       0
#XS Ineff= 2 , 0
          389.69 1211.43
Permanent Ineff=
       F       F
Bank Sta=452.3,467.3
XS Rating Curve= 0 ,0
Exp/Cntr=0.3,0.1

Type RM Length L Ch R = 1 ,9871.4  ,368.5,367.9,367.3
XS GIS Cut Line= 2
     1743688.412      278000.865     1743378.926      278463.181
#Sta/Elev= 30
       0 1263.64     9.8 1253.54    19.5 1249.36    29.3 1243.45      39 1234.93
    58.6 1220.86    78.1 1210.67    87.8 1206.92    97.6 1204.52   117.1 1201.09
   126.9 1200.44   136.6 1200.64   185.4 1204.84   214.7  1205.2   224.5 1203.82
   253.8 1196.73   312.3 1196.61   322.1 1195.95   341.6 1193.02   348.3  1193.4
   351.4 1193.58   363.3 1198.34   380.7    1207   390.4 1208.13   400.2 1212.63
   419.7 1224.13   458.7 1245.43   478.3 1251.35   517.3 1273.21   556.3 1297.72
#Mann= 3 , 0 , 0
       0     .08       0   348.3    .045       0   363.3     .08       0
Bank Sta=348.3,363.3
XS Rating Curve= 0 ,0
Exp/Cntr=0.3,0.1

Type RM Length L Ch R = 1 ,9503.3  ,390.5,385,379.4
XS GIS Cut Line= 2
     1743349.551      277852.375     1743090.824      278267.111
#Sta/Elev= 30
       0 1276.28    39.1 1256.34    58.7  1244.9    68.4 1243.35    78.2 1239.66
   136.9 1209.89   146.6 1207.25   166.2 1206.25     176 1203.81   185.8 1198.98
   205.3 1185.67   215.1 1183.27   224.9 1183.17   225.8 1183.23   240.8  1184.3
     264 1185.43   312.8 1189.49   322.6 1191.81   342.2 1201.03     352 1204.46
   371.5 1223.64   391.1 1236.28   410.6 1246.27   420.4 1250.24   430.2  1251.1
   439.9 1255.69   449.7 1261.55   459.5 1269.52   469.3 1279.03   488.8  1299.5
#Mann= 3 , 0 , 0
       0     .08       0   225.8    .045       0   240.8     .08       0
Bank Sta=225.8,240.8
XS Rating Curve= 0 ,0
Exp/Cntr=0.3,0.1

Type RM Length L Ch R = 1 ,9118.2  ,407.3,407,406.7
XS GIS Cut Line= 2
     1742959.641      277727.079     1742852.128      278070.716
#Sta/Elev= 30
       0 1249.78     9.7 1248.67    29.2 1235.26    58.4 1215.97    77.8 1201.45
    87.6 1199.05    97.3 1197.26     107  1196.1   116.8 1195.12   126.5 1192.52
   136.2 1188.68     146 1184.38   155.7 1180.75   165.4 1179.23   173.9 1179.25
   184.9 1179.91   188.9 1180.71   204.4 1183.81   233.6 1189.07   243.3  1190.4
   262.8  1191.1   272.5 1192.53   282.2 1196.78   291.9  1203.2   311.4  1216.6
   321.1 1224.88   330.9 1231.75   340.6 1235.35   350.3 1242.72   360.1 1249.42
#Mann= 3 , 0 , 0
       0     .08       0   173.9    .045       0   188.9     .08       0
Bank Sta=173.9,188.9
XS Rating Curve= 0 ,0
Exp/Cntr=0.3,0.1

Type RM Length L Ch R = 1 ,8711.1  ,398.6,399.9,401.2
XS GIS Cut Line= 2
     1742569.266      277612.608     1742454.026      277992.737
#Sta/Elev= 30
       0 1221.11     9.7 1216.13    19.4 1213.15    29.1 1211.17    67.8 1194.91
    87.2  1185.8    96.9 1182.99   116.3 1182.25     126 1181.59   135.6 1179.87
   145.3 1177.33   164.7 1171.41   174.4 1170.27   184.1 1170.28   188.8 1170.83
   193.8 1171.41   203.8 1173.97   213.1 1176.35   222.8 1178.36   232.5  1180.2
   242.2 1181.39   251.9 1181.75   271.3 1181.89   300.3 1183.43   319.7 1184.75
   339.1 1187.47   348.8 1190.84   358.5 1197.93   368.2 1205.41   397.2 1228.87
#Mann= 3 , 0 , 0
       0     .08       0   188.8    .045       0   203.8     .08       0
Bank Sta=188.8,203.8
XS Rating Curve= 0 ,0
Exp/Cntr=0.3,0.1

Type RM Length L Ch R = 1 ,8311.1  ,395.4,400,404.6
XS GIS Cut Line= 2
     1742198.456      277503.516     1742078.617        277827.9
#Sta/Elev= 30
       0  1206.4     9.6 1198.48    19.2 1192.62    28.8 1190.29    38.4  1182.7
      48  1176.6    57.6 1172.55    67.2 1171.08    86.4 1171.03   105.7 1171.45
   124.9 1171.25   134.5 1169.44   144.1 1165.11   153.7 1162.27   163.3 1163.22
   168.3 1165.43   172.9 1167.47   182.5 1172.11   183.3 1172.17   192.1 1172.87
   201.7  1175.5   211.3 1178.93   220.9 1181.55   230.5 1182.98   240.2 1183.33
   278.6 1183.25   288.2 1185.04   326.6 1196.81   336.2 1200.76   345.8 1205.54
#Mann= 3 , 0 , 0
       0     .08       0   168.3    .045       0   183.3     .08       0
Bank Sta=168.3,183.3
XS Rating Curve= 0 ,0
Exp/Cntr=0.3,0.1

Type RM Length L Ch R = 1 ,7911.1  ,394.7,399.8,404.9
XS GIS Cut Line= 2
     1741879.382      277335.213     1741695.762      277629.858
#Sta/Elev= 30
       0 1213.43     9.6 1209.19    19.3 1207.97    28.9 1202.68    48.2 1191.77
    57.9 1186.45    67.5 1182.54    96.4 1174.24   115.7 1171.25     135 1165.67
   144.7 1163.08   154.3 1160.85   163.9 1158.47   173.6 1155.89   180.3 1154.75
   183.2 1154.25   195.3 1154.45   202.5 1154.63   221.8 1157.91   231.4  1159.3
   241.1  1161.1   250.7 1164.22   260.4 1168.32   279.7 1176.67   289.3 1179.76
     299 1181.27   308.6 1184.58   318.2 1186.21   327.9 1187.13   347.2 1188.53
#Mann= 3 , 0 , 0
       0     .08       0   180.3    .045       0   195.3     .08       0
Bank Sta=180.3,195.3
XS Rating Curve= 0 ,0
Exp/Cntr=0.3,0.1

Type RM Length L Ch R = 1 ,7511.1  ,398.1,400,402
XS GIS Cut Line= 2
     1741609.809      277104.925     1741341.458      277374.221
#Sta/Elev= 30
       0 1190.86     9.8 1186.76    19.5 1183.01      78 1161.32    87.7 1158.45
    97.5 1155.06   107.2 1152.82     117 1153.45   126.7 1154.77   136.5 1154.89
   146.2 1153.85     156 1152.42   165.7 1150.92   185.2 1147.47     195 1146.71
   195.4 1146.71   204.7 1146.76   210.4 1147.35   214.5 1147.78     234 1153.85
   243.7 1158.26   282.7 1179.63   292.4  1184.6   302.2 1187.51   311.9 1188.72
   331.4 1192.87   341.2 1197.72   350.9 1206.04   360.7 1211.98   380.2 1222.44
#Mann= 3 , 0 , 0
       0     .08       0   195.4    .045       0   210.4     .08       0
Bank Sta=195.4,210.4
XS Rating Curve= 0 ,0
Exp/Cntr=0.3,0.1

Type RM Length L Ch R = 1 ,7111.1  ,402.2,399.9,397.7
XS GIS Cut Line= 2
     1741421.458      276765.999     1741071.529      277062.094
#Sta/Elev= 30
       0  1204.8     9.8 1197.72    19.5 1191.42   107.3  1162.8     117 1159.94
   136.5 1152.13     156 1145.67   165.8 1143.32   175.6 1142.84   195.1 1145.12
   204.8 1145.65   214.6 1144.72   234.1 1142.14   243.8 1139.72   247.9 1139.62
   253.6 1139.49   262.9 1141.57   282.8 1147.48   292.6 1151.39   302.3 1156.08
   341.4 1175.86   351.1 1178.83   360.9 1184.16   370.6 1189.18   380.4  1193.5
   409.6 1207.78   419.4  1212.8   438.9 1224.08   448.6 1229.45   458.4 1231.33
#Mann= 3 , 0 , 0
       0     .08       0   247.9    .045       0   262.9     .08       0
#XS Ineff= 2 , 0
          205.04 1145.49
Permanent Ineff=
       F       F
Bank Sta=247.9,262.9
XS Rating Curve= 0 ,0
Exp/Cntr=0.3,0.1

Type RM Length L Ch R = 1 ,6711.1  ,401.6,401.1,399.8
XS GIS Cut Line= 2
      1741131.18      276458.048     1740802.839      276798.329
#Sta/Elev= 30
       0 1243.75    38.6 1217.59    48.2 1208.88    57.9 1201.49    67.6 1195.95
    77.2 1193.68    86.8 1188.03   135.1 1156.01   154.4 1144.14     164 1139.64
   173.7 1139.37   183.4 1140.29     193 1140.86   202.7 1140.09   212.3 1137.39
     222 1134.18   231.6    1132   234.3 1131.88   241.3 1131.56   249.3 1131.96
   270.2 1134.18   279.9 1134.52   289.5 1135.25   318.5 1139.38   347.4 1144.29
   376.4 1150.54   424.6 1155.78   434.3 1157.23   453.6 1158.66   472.9 1160.44
#Mann= 3 , 0 , 0
       0     .08       0   234.3    .045       0   249.3     .08       0
Bank Sta=234.3,249.3
XS Rating Curve= 0 ,0
Exp/Cntr=0.3,0.1

Type RM Length L Ch R = 1 ,6309.8  ,417.3,409.8,403.1
XS GIS Cut Line= 2
     1740832.774      276222.056     1740496.546      276573.854
#Sta/Elev= 30
       0 1195.04     9.7 1192.36    19.5 1188.12    38.9 1178.53    48.7 1176.06
    58.4 1168.64    68.1 1162.08    97.3 1145.68   107.1 1140.56   116.8 1136.39
   126.5 1134.85   155.7 1135.46   175.2 1134.55   194.6 1131.83   269.8 1124.32
   282.2 1124.04   284.8 1124.54     292 1125.92   301.7 1131.21   321.2 1148.48
   350.4 1165.06   360.1 1168.36   369.8 1173.05     399 1190.73   428.2 1207.44
     438 1214.67   447.7 1222.83   457.4 1228.55   476.9 1235.85   486.6 1241.59
#Mann= 3 , 0 , 0
       0     .08       0   269.8    .045       0   284.8     .08       0
Bank Sta=269.8,284.8
XS Rating Curve= 0 ,0
Exp/Cntr=0.3,0.1

Type RM Length L Ch R = 1 ,5898.8  ,386.7,393.7,400.7
XS GIS Cut Line= 2
     1740473.203      275890.529     1740274.953      276347.085
#Sta/Elev= 30
       0 1138.88     9.8  1134.4    19.5 1131.75    29.3 1130.61    58.6 1129.54
    68.3 1129.37    97.6 1129.33   126.9 1128.98   185.4 1128.86     205  1127.2
   214.7 1125.95   254.9  1119.9   263.5 1119.08   269.9 1119.82   273.3 1120.22
     283 1122.34   292.8 1126.11   302.6 1132.89   312.3 1138.72   351.4 1160.21
   361.1 1164.51   370.9 1165.89   390.4 1176.88   409.9 1189.16   419.7 1195.03
   439.2 1205.92   448.9 1209.46   458.7 1212.02   478.2 1223.16   497.7 1233.78
#Mann= 3 , 0 , 0
       0     .08       0   254.9    .045       0   269.9     .08       0
Bank Sta=254.9,269.9
XS Rating Curve= 0 ,0
Exp/Cntr=0.3,0.1

Type RM Length L Ch R = 1 ,5504.9  ,414.6,400.5,386.3
XS GIS Cut Line= 2
     1740224.521      275731.921     1739911.299      276090.717
#Sta/Elev= 30
       0 1196.53    19.4 1196.07    29.2 1194.89    38.9 1190.51      68 1166.36
    77.8 1155.14    87.5 1145.59    97.2 1138.33   106.9 1131.74   116.6  1127.6
   126.4 1125.27   136.1 1121.49   165.2 1117.74   184.7 1117.56   233.3 1123.52
   272.2 1129.84   281.9 1128.82   291.6 1124.08   301.3 1117.22     311 1112.02
   318.9 1110.67   330.5 1109.76   333.9 1112.43   340.2 1117.38   349.9 1128.95
   359.6 1137.45   408.2 1177.34   427.7 1186.27   456.8 1207.72   476.3 1225.41
#Mann= 3 , 0 , 0
       0     .08       0   318.9    .045       0   333.9     .08       0
Bank Sta=318.9,333.9
XS Rating Curve= 0 ,0
Exp/Cntr=0.3,0.1

Type RM Length L Ch R = 1 ,5104.2  ,329.5,320.1,310.7
XS GIS Cut Line= 2
     1739753.294      275516.368     1739716.884      275916.894
#Sta/Elev= 30
       0  1119.4     9.8 1115.62    19.6 1113.34    29.4 1112.31    88.3 1110.99
   107.9 1109.87   127.5 1109.26     157  1107.7   166.8 1106.84   176.6 1104.08
   182.5 1101.76   186.4 1100.22   196.2 1098.44   197.5 1098.46     206 1098.57
   215.8 1100.75   225.6 1107.96     255 1140.69   264.8 1153.37   274.7 1163.84
   284.5 1168.63   294.3 1180.03   304.1 1185.98   313.9 1187.67   333.5 1187.78
   343.3 1188.81   353.1 1190.28   362.9 1190.84   372.8 1193.15   402.2 1201.14
#Mann= 3 , 0 , 0
       0     .08       0   182.5    .045       0   197.5     .08       0
Bank Sta=182.5,197.5
XS Rating Curve= 0 ,0
Exp/Cntr=0.3,0.1

Type RM Length L Ch R = 1 ,4784.1  ,447.3,465.9,484.4
XS GIS Cut Line= 2
     1739357.394      275576.569     1739496.897      275989.314
#Sta/Elev= 30
       0 1171.79     9.7 1164.57    19.4 1156.16      29 1146.49    38.7 1139.71
    48.4  1134.8    58.1 1125.01    67.8 1116.71    77.4  1110.4    87.1  1106.4
    96.8 1104.22   106.5 1103.05   135.6 1102.65   154.9 1103.53   164.6 1102.75
     184 1099.94   203.3 1098.79     213 1095.58   222.7 1094.89   226.6 1093.77
   232.4  1092.1   241.6 1092.75   261.4 1099.61   290.5 1106.07   309.8 1109.69
   319.5  1114.6   377.6 1152.52   387.3 1153.46   416.3 1173.07   435.7 1183.15
#Mann= 3 , 0 , 0
       0     .08       0   226.6    .045       0   241.6     .08       0
Bank Sta=226.6,241.6
XS Rating Curve= 0 ,0
Exp/Cntr=0.3,0.1

Type RM Length L Ch R = 1 ,4317.8  ,223.4,228.9,234.4
XS GIS Cut Line= 3
     1739083.864      275561.783      1738872.28      275953.969
      1738865.65      275966.258
#Sta/Elev= 30
       0 1133.86     9.7 1128.83    29.1  1117.6    38.8  1114.3    48.4 1109.94
    67.8 1098.73    77.5 1095.12    87.2 1094.41   106.6 1094.35   125.9 1093.08
   145.3 1091.08   174.4 1089.52   193.8 1083.08   201.1 1082.12   203.4 1081.82
   216.1 1082.85   222.8 1083.34   232.5 1087.23   242.2 1089.48   271.2 1090.42
     310 1090.69   319.7 1092.88   329.4 1099.28   377.8 1137.67   387.5 1139.78
   397.2 1146.44   416.6 1161.49   426.2  1167.9   445.6 1179.29   459.6 1188.17
#Mann= 3 , 0 , 0
       0     .08       0   201.1    .045       0   216.1     .08       0
Bank Sta=201.1,216.1
XS Rating Curve= 0 ,0
Exp/Cntr=0.3,0.1

Type RM Length L Ch R = 1 ,4089    ,540.3,527.1,513.9
XS GIS Cut Line= 2
     1738957.766      275439.097     1738641.021      275787.647
#Sta/Elev= 30
       0 1122.37     9.8 1118.52    39.2 1103.74    58.9 1095.71    68.7 1092.68
    78.5 1091.08    88.3 1090.29   166.8 1085.12   186.4 1084.99   196.2 1084.05
     206 1081.31   210.8 1079.06   215.9 1076.67   225.8 1079.24   245.3 1089.44
   294.4 1110.04   304.2 1115.71   323.8 1130.88   333.6 1142.01   343.4 1149.02
   353.2 1154.03     363 1158.42   372.8 1161.94   382.7 1164.36   392.5 1165.54
   402.3 1165.38   441.5 1167.13   451.4 1168.45   461.2 1170.81     471 1173.89
#Mann= 3 , 0 , 0
       0     .08       0   210.8    .045       0   225.8     .08       0
Bank Sta=210.8,225.8
XS Rating Curve= 0 ,0
Exp/Cntr=0.3,0.1

Type RM Length L Ch R = 1 ,3561.9  ,480.8,490.3,499.8
XS GIS Cut Line= 3
     1738341.206      275276.844     1738285.816      275634.338
     1738284.827      275640.717
#Sta/Elev= 30
       0 1130.11    19.6 1117.87    29.3 1111.42    39.1 1105.74    48.9 1104.95
    78.2 1084.48      88 1078.44    97.8 1075.13   107.6  1073.4   127.1 1073.13
   136.9 1074.15   146.7 1074.52   156.4 1070.11   166.2 1065.17   166.5 1065.14
     176  1064.3   181.5 1065.99   185.8 1067.32   195.6 1071.91   205.3 1072.66
   215.1 1074.09   224.9 1074.39     264 1074.16   273.8 1074.88   283.5 1075.21
   293.3 1077.51   322.6 1088.81     352 1099.65   361.8 1101.13   368.2 1101.86
#Mann= 3 , 0 , 0
       0     .08       0   166.5    .045       0   181.5     .08       0
Bank Sta=166.5,181.5
XS Rating Curve= 0 ,0
Exp/Cntr=0.3,0.1

Type RM Length L Ch R = 1 ,3071.6  ,363,360.9,358.8
XS GIS Cut Line= 2
     1737959.699      275150.815     1737748.941      275476.842
#Sta/Elev= 30
       0 1112.42    19.4 1099.39    29.1 1093.91    38.8 1089.19    67.9 1077.39
    77.6 1074.64    87.4 1070.19      97 1067.09   116.5 1063.94   135.9 1061.68
   145.6 1063.21   155.3 1062.59     165 1060.58   179.9 1056.24   184.4 1054.82
   194.9 1055.73   223.2 1061.97   232.9 1062.77     262 1062.69   271.8 1063.48
   281.5  1066.8   291.2 1071.66   300.9 1075.39   310.6 1076.02   320.3 1075.94
     330 1076.42   349.4  1078.2   368.8 1082.58   378.5 1085.42   388.2  1089.6
#Mann= 3 , 0 , 0
       0     .08       0   179.9    .045       0   194.9     .08       0
Bank Sta=179.9,194.9
XS Rating Curve= 0 ,0
Exp/Cntr=0.3,0.1

Type RM Length L Ch R = 1 ,2710.4  ,391.5,378,364.4
XS GIS Cut Line= 2
     1737631.201      274975.577     1737455.209      275309.818
#Sta/Elev= 30
       0 1066.79     9.7  1062.7    19.4  1059.9    29.1 1058.67    38.7 1058.38
    58.1  1057.2    87.2 1056.28    96.9 1056.52   106.5 1056.46   116.2 1053.31
   125.9 1048.59     134 1047.64   135.6 1047.45     149  1048.9   164.7 1050.76
   193.7 1057.06   213.1 1058.09   222.8 1060.66   232.5 1065.18   242.1 1068.54
   251.8 1070.62   271.2 1081.92   280.9 1087.35   309.9 1102.62   319.6 1106.35
   329.3 1108.55   348.7 1119.12   358.4 1125.12   368.1 1131.78   377.7 1137.62
#Mann= 3 , 0 , 0
       0     .08       0     134    .045       0     149     .08       0
Bank Sta=134,149
XS Rating Curve= 0 ,0
Exp/Cntr=0.3,0.1

Type RM Length L Ch R = 1 ,2332.5  ,424.1,426.8,429.5
XS GIS Cut Line= 2
     1737182.494      274927.173     1737225.469      275296.483
#Sta/Elev= 29
       0 1058.38     9.8 1057.43    19.6 1055.38    39.1 1050.78    48.9 1049.21
    58.7  1048.8    97.8 1049.85   117.4  1050.6   156.6 1052.29   166.3 1052.49
   176.1 1050.89     194 1041.61   195.7 1040.72   205.5 1039.76     209 1040.45
   215.2 1041.68   234.8 1046.98   244.6 1048.76   254.4 1050.96   264.2 1057.73
   283.7 1074.16   303.3 1090.38   313.1 1098.64   322.9 1104.77   332.7 1107.11
   342.4 1115.66   352.2 1124.09     362 1132.06   371.8 1138.45
#Mann= 3 , 0 , 0
       0     .08       0     194    .045       0     209     .08       0
Bank Sta=194,209
XS Rating Curve= 0 ,0
Exp/Cntr=0.3,0.1

Type RM Length L Ch R = 1 ,1905.6  ,511.1,512,512.9
XS GIS Cut Line= 2
     1736780.973      274950.104      1736779.94      275313.935
#Sta/Elev= 30
       0 1053.72    19.7 1047.56    29.5  1044.9    39.3 1044.88    49.2 1043.18
      59 1042.28    78.7 1041.59   108.2 1038.69     118 1038.68   137.7 1036.61
   147.5 1036.76   157.3 1039.72   167.2 1041.66     177 1036.64   186.8 1030.69
   193.8 1030.68   196.7 1030.67   206.5    1029   208.8  1029.2   216.3 1029.87
     236 1033.77   255.7 1037.03   265.5 1040.42   275.3 1040.46   285.2 1046.35
   324.5  1071.2   334.3 1078.99   344.2 1086.07     354  1086.2   363.8 1093.51
#Mann= 3 , 0 , 0
       0     .08       0   193.8    .045       0   208.8     .08       0
#XS Ineff= 2 , 0
          167.24  1041.5
Permanent Ineff=
       F       F
Bank Sta=193.8,208.8
XS Rating Curve= 0 ,0
Exp/Cntr=0.3,0.1

Type RM Length L Ch R = 1 ,1393.4  ,440.9,442.3,443.8
XS GIS Cut Line= 2
     1736280.925      274958.334      1736264.76      275313.935
#Sta/Elev= 30
       0 1044.42     9.6  1039.3    19.2 1036.43    28.9 1035.78    67.4  1034.2
    86.6 1033.81   144.3 1031.11   153.9 1030.86   163.6 1029.17   173.2  1025.3
   175.8 1024.64   182.8 1022.86   190.8 1023.46   192.4 1023.58     202 1025.94
   211.7 1028.48   221.3 1030.14   230.9 1030.95   240.5 1031.23   250.1 1032.36
   259.8 1034.16   269.4 1037.95   288.6 1047.98   298.2 1053.25   307.9 1058.06
   317.5 1058.47   327.1 1064.04   336.7 1070.14   346.4 1076.63     356 1082.76
#Mann= 3 , 0 , 0
       0     .08       0   175.8    .045       0   190.8     .08       0
Bank Sta=175.8,190.8
XS Rating Curve= 0 ,0
Exp/Cntr=0.3,0.1

Type RM Length L Ch R = 1 ,951.1   ,317.3,319.5,321.6
XS GIS Cut Line= 2
     1735849.775      274962.334     1735807.794      275343.306
#Sta/Elev= 30
       0 1051.87     9.8 1047.92    29.5  1040.2    39.3 1037.06    49.1 1036.08
      59 1031.76    68.8 1028.42    78.6 1027.31    88.4 1027.26   127.8 1026.67
   137.6 1025.74   147.4 1021.98   154.6 1018.39   157.2 1017.09   167.1 1016.12
   169.6 1016.69   176.9 1018.37   186.7 1021.44   196.6 1022.69   206.4 1022.71
   216.2 1022.96   275.2 1023.64     285 1023.62   314.5 1023.89   334.1 1023.61
     344 1024.78   353.8 1029.06   363.6 1028.94   373.4 1034.46   383.3 1040.33
#Mann= 3 , 0 , 0
       0     .08       0   154.6    .045       0   169.6     .08       0
Bank Sta=154.6,169.6
XS Rating Curve= 0 ,0
Exp/Cntr=0.3,0.1

Type RM Length L Ch R = 1 ,631.6   ,101.8,92.1,82.2
XS GIS Cut Line= 2
     1735552.975      274900.365     1735449.911      275395.077
#Sta/Elev= 30
       0 1089.95     9.7 1089.54    19.4 1081.64    48.6  1056.7    77.7    1033
    87.5 1030.38   106.9  1022.6   116.6 1021.36     136 1020.29   145.8 1017.95
   155.5 1012.84   163.7    1010   165.2 1009.48   174.9 1009.14   178.7 1009.27
   184.6 1009.48   204.1 1013.26   213.8 1014.48     243 1015.43     311 1016.32
   330.4 1017.15   340.1 1020.26   388.7 1047.02   398.4  1052.9   408.2 1056.07
   417.9 1060.41   427.6 1067.99   485.9 1115.68   495.6 1121.06   505.3 1128.13
#Mann= 3 , 0 , 0
       0     .08       0   163.7    .045       0   178.7     .08       0
Bank Sta=163.7,178.7
XS Rating Curve= 0 ,0
Exp/Cntr=0.3,0.1

Type RM Length L Ch R = 1 ,539.5   ,548.5,539.3,530.4
XS GIS Cut Line= 4
     1735445.778      274877.983     1735417.754      275013.136
     1735461.773      275206.126      1735427.34      275394.136
#Sta/Elev= 30
       0 1085.58    18.4 1071.17    27.6 1067.15    36.8 1064.15    55.2 1050.29
      92 1024.76   101.2 1020.39   156.9 1014.98   172.9 1008.87   175.7 1007.69
   185.2 1006.68   187.9 1006.68     204 1007.55   222.9  1010.7   241.7 1012.84
   317.1  1015.2   326.6 1016.59     336 1019.68   345.5  1025.6   355.1 1026.32
   374.2 1038.15   402.9 1054.89     422 1070.57   441.1  1077.8   460.2 1091.21
   488.9 1114.77   498.4 1121.98     508 1127.42   517.6 1129.15   527.1    1136
#Mann= 3 , 0 , 0
       0     .08       0   172.9    .045       0   187.9     .08       0
Bank Sta=172.9,187.9
XS Rating Curve= 0 ,0
Exp/Cntr=0.3,0.1

Chan Stop Cuts=-1
Use User Specified Reach Order=0
Composite Channel Slope=5
